--- ShinsRn.prj (project) ---

Proj Title=ShinsRn
Current Plan=p01
Default Exp/Contr=0,0
English Units
Geom File=g01
Flow File=f01
Plan File=p01
BEGIN DESCRIPTION:
END DESCRIPTION:
DSS Export Rating Curves= 0
DSS Export Rating Curve Sorted= 0
DSS Export Volume Flow Curves= 0
DXF OffsetX= 0
DXF OffsetY= 0
DXF ScaleX= 0
DXF ScaleY= 0

--- ShinsRn.p01 (plan) ---

Plan Title=Floodplain
Program Version=4.00
Geom File=g01
Flow File=f01
K Sum by GR=0
Std Step Tol=0.01
Critical Tol=0.01
Num of Std Step Trials=20
Max Error Tol=0.3
Flow Tol Ratio=0.001
Split Flow NTrial=30
Split Flow Tol=0.02
Split Flow Ratio=0.02
Log Output Level=0
Friction Slope Method=1
Unsteady Friction Slope Method=2
Unsteady Bridges Friction Slope Method=1
Global Log Level=0
CheckData=False
Run HTab=0
Run UNet=0
Run PostProcess=0
UNET Theta=0
UNET Theta Warmup=0
UNET ZTol=0
UNET ZSATol=0
UNET MxIter=0
UNET MaxInSteps=0
UNET DtIC=0
UNET DtMin=0
UNET MaxCRTS=0
UNET WFStab=0
UNET SFStab=0
UNET WFX=0
UNET SFX=0
UNET DSS MLevel=0
UNET DZMax Abort=0
UNET Convert EG Bridges=0
UNET Use Existing IB Tables=0
UNET Froude Limit=0
UNET Froude Power=0
Write IC File=0
Echo Input=False
Echo Output=False
Write Detailed=0

--- ShinsRn.f01 (steady flow) ---

Flow Title=NFF Regression Equation
Program Version=4.00
Number of Profiles= 1
Profile Names=P100yr
River Rch & RM=ShinsRn,Main            ,27629.1
717.7026
River Rch & RM=ShinsRn,Main            ,27311.6
847.6105
River Rch & RM=ShinsRn,Main            ,25593.4
900.3053
River Rch & RM=ShinsRn,Main            ,23908.7
 999.854
River Rch & RM=ShinsRn,Main            ,22029.1
1070.265
River Rch & RM=ShinsRn,Main            ,19229.1
1168.782
River Rch & RM=ShinsRn,Main            ,18829.1
1402.994
River Rch & RM=ShinsRn,Main            ,16829.1
1432.737
River Rch & RM=ShinsRn,Main            ,16429.1
1738.446
River Rch & RM=ShinsRn,Main            ,15318.2
1794.289
River Rch & RM=ShinsRn,Main            ,11329
1983.229
River Rch & RM=ShinsRn,Main            ,6029.1
2192.858
River Rch & RM=ShinsRn,Main            ,29.1
2408.466
River Rch & RM=ShinsRn,Main            ,29.1
2412.229
Boundary for River Rch & Prof#=ShinsRn,Main            , 1
Up Type= 0
Dn Type= 1
Dn Known WS=913.43
DSS Import GetInterval= 0
DSS Import GetPeak= 0
DSS Import FillOption= 0

--- ShinsRn.g01 (geometry) ---

Geom Title=USGS 3m DEM
Program Version=4.00

River Reach=ShinsRn     ,Main
Reach XY= 30
     1756473.384      309025.720     1755583.496      309080.455
     1754993.508      309658.871     1753526.575      309754.920
     1752121.859      310672.011     1751432.035      312208.409
     1751575.038      312367.096     1751352.675      312796.231
     1751482.232      313008.086     1751233.586      313596.546
     1751228.563      314505.658     1750504.317      315212.305
     1749362.608      315812.274     1749221.991      316532.507
     1748960.558      316400.530     1748719.858      316702.342
     1748578.677      317464.165     1747415.125      318199.900
     1747498.111      319703.183     1747112.407      319873.134
     1746636.003      320738.912     1745718.984      321143.424
     1745438.872      321702.501     1744640.043      322445.288
     1743020.450      322088.052     1742826.344      322396.486
     1742343.947      322438.035     1742156.215      322789.527
     1742666.852      323816.514     1742283.457      325032.518

Type RM Length L Ch R = 1 ,27629.1,311.996,317.517,317.644
XS GIS Cut Line= 3
     1756348.134      308541.311     1756463.386      309025.911
     1756472.955      309526.320
#Sta/Elev= 30
       0 1122.42   128.2 1108.05   170.8 1105.59   177.0 1104.78   181.8 1103.81
   201.4 1096.08   261.8 1076.40   284.6 1068.25   299.7 1064.82   311.3 1063.36
   335.7 1061.30   460.1 1056.34   482.3 1054.72   490.6 1054.54   504.2 1054.24
   505.6 1054.31   546.5 1056.44   647.5 1060.66   654.4 1061.10   688.4 1065.61
   718.0 1074.64   750.5 1086.55   765.0 1090.17   805.7 1098.41   853.6 1105.95
   895.5 1113.44   918.8 1118.15   952.4 1123.07   968.1 1125.94   998.6 1129.91
#Mann= 3 , 0 , 0
       0     0.1       0   490.6   0.045       0   505.6     0.1       0
Bank Sta=   490.6,   505.6
Exp/Cntr=0.3,0.1

Type RM Length L Ch R = 1 ,27311.6,488.23,482.483,480.04
XS GIS Cut Line= 3
     1756150.555      308531.560     1756146.182      309048.443
     1756160.147      309546.554
#Sta/Elev= 30
       0 1186.60    40.0 1185.44    61.4 1181.65   110.7 1169.41   130.3 1164.17
   156.3 1158.00   193.3 1150.50   274.2 1127.20   336.3 1107.48   357.0 1099.17
   391.6 1085.99   439.3 1067.27   453.8 1061.99   466.9 1056.76   474.9 1054.06
   489.5 1050.93   500.4 1050.31   509.6 1050.10   515.4 1050.44   588.2 1054.59
   747.3 1064.21   781.7 1069.20   826.1 1076.36   862.3 1084.99   890.0 1090.27
   908.3 1092.92   930.1 1094.55   970.7 1096.63  1006.0 1101.63  1015.2 1103.67
#Mann= 3 , 0 , 0
       0     0.1       0   500.4   0.045       0   515.4     0.1       0
Bank Sta=   500.4,   515.4
Exp/Cntr=0.3,0.1

Type RM Length L Ch R = 1 ,26829.1,347.092,336.709,327.271
XS GIS Cut Line= 3
     1755591.292      308568.219     1755691.806      309058.535
     1755807.788      309545.539
#Sta/Elev= 30
       0 1140.56     3.2 1141.03    16.5 1140.69    78.6 1133.90   116.3 1130.69
   135.6 1128.80   184.7 1121.48   238.7 1117.03   292.4 1110.39   301.1 1108.90
   328.6 1102.34   338.9 1099.29   442.5 1071.57   466.2 1061.54   487.7 1050.20
     493 1048.67   501.7 1046.10     508 1046.20   595.0 1047.58   693.9 1047.33
   781.2 1052.56   797.4 1057.55   811.3 1063.47   823.9 1064.93   836.0 1066.72
   864.1 1074.40   873.7 1077.60   915.2 1090.61   951.4 1097.23  1001.1 1103.85
#Mann= 3 , 0 , 0
       0     0.1       0     493   0.045       0     508     0.1       0
Bank Sta=     493,     508
Exp/Cntr=0.3,0.1

Type RM Length L Ch R = 1 ,26492.4,461.365,463.291,459.95
XS GIS Cut Line= 3
     1755097.555      308796.947     1755404.111      309203.675
     1755698.792      309604.023
#Sta/Elev= 30
       0 1168.84     6.5 1168.52    36.3 1170.25    64.4 1167.25    79.3 1163.82
    96.7 1157.24   118.6 1151.24   243.1 1121.70   311.4 1106.79   361.8 1092.75
   434.0 1068.33   494.8 1043.79   499.9 1043.18   505.9 1042.46   514.9 1042.81
   552.1 1044.92   611.5 1045.36   696.8 1048.27   726.8 1050.52   755.8 1051.31
   775.0 1053.77   800.0 1059.18   818.1 1061.54   837.1 1062.41   877.4 1070.16
   901.8 1076.23   930.5 1081.00   971.2 1089.39   986.9 1091.48  1006.4 1095.20
#Mann= 3 , 0 , 0
       0     0.1       0   499.9   0.045       0   514.9     0.1       0
Bank Sta=   499.9,   514.9
Exp/Cntr=0.3,0.1

Type RM Length L Ch R = 1 ,26029.1,422.857,435.751,448.714
XS GIS Cut Line= 3
     1754812.026      309063.681     1755110.080      309534.797
     1755456.578      309881.914
#Sta/Elev= 30
       0 1128.40    19.0 1124.50    55.1 1118.23    63.3 1116.10   127.6 1102.29
   157.1 1095.47   188.6 1087.01   196.3 1084.04   252.4 1059.55   271.7 1056.82
   302.9 1054.59   394.1 1049.14     550 1040.63   559.7 1040.11     565 1040.46
   621.7 1045.58   637.0 1050.40   659.9 1060.78   676.6 1065.27   699.0 1067.56
   768.9 1084.73   797.2 1092.36   867.6 1106.65   874.6 1107.78   981.2 1118.88
  1014.2 1121.65  1023.2 1120.72  1028.4 1120.81  1045.9 1117.22  1047.9 1117.16
#Mann= 3 , 0 , 0
       0     0.1       0     550   0.045       0     565     0.1       0
Bank Sta=     550,     565
Exp/Cntr=0.3,0.1

Type RM Length L Ch R = 1 ,25593.4,365.221,364.249,369.917
XS GIS Cut Line= 3
     1754719.146      309093.025     1754744.842      309587.474
     1754893.410      310122.937
#Sta/Elev= 30
       0 1119.17    37.7 1105.49    64.1 1095.06   108.0 1080.97   131.2 1076.67
   166.9 1076.02   178.8 1073.67   187.7 1070.83   221.6 1060.95   226.3 1059.98
   262.0 1057.37   303.8 1053.17   359.4 1048.24   487.2 1037.41   487.9 1037.35
   502.2 1038.12   508.6 1038.49   528.9 1042.90   542.5 1045.30   598.2 1053.10
   658.6 1060.07   693.4 1062.57   751.7 1072.21   772.9 1074.15   830.7 1077.36
   841.5 1078.32   900.9 1081.02   969.3 1083.17  1013.5 1083.88  1050.8 1083.67
#Mann= 3 , 0 , 0
       0     0.1       0   487.2   0.045       0   502.2     0.1       0
Bank Sta=   487.2,   502.2
Exp/Cntr=0.3,0.1

Type RM Length L Ch R = 1 ,25229.1,400.111,400,396.326
XS GIS Cut Line= 3
     1754352.777      309194.348     1754399.652      309694.464
     1754407.866      310194.578
#Sta/Elev= 30
       0 1126.62    14.1 1121.63    53.7 1109.96    83.7 1098.65   101.4 1089.71
   113.3 1086.68   128.7 1086.80   144.9 1088.82   164.4 1087.85   188.4 1085.65
   229.6 1078.07   277.3 1067.90   288.1 1063.68   321.4 1048.66   337.7 1047.17
   351.8 1044.48   380.8 1041.65   494.8 1033.69   506.8 1033.07   509.8 1033.38
   563.8 1039.49   585.1 1040.78   614.9 1047.39   628.3 1049.62   653.8 1050.68
   717.3 1056.17   815.5 1075.42   890.5 1086.71   929.9 1096.47  1002.5 1109.81
#Mann= 3 , 0 , 0
       0     0.1       0   494.8   0.045       0   509.8     0.1       0
Bank Sta=   494.8,   509.8
Exp/Cntr=0.3,0.1

Type RM Length L Ch R = 1 ,24829.1,507.234,507.01,501.074
XS GIS Cut Line= 3
     1753951.165      309208.094     1754000.277      309706.146
     1754101.049      310262.219
#Sta/Elev= 30
       0 1161.86    54.8 1167.11   106.4 1169.63   142.0 1170.87   158.5 1168.95
   180.3 1162.14   242.7 1134.69   266.6 1128.82   290.4 1114.23   297.6 1111.22
   302.4 1108.48   307.5 1107.81   318.2 1104.33   342.6 1100.55   375.7 1092.83
   385.9 1087.68   398.2 1080.38   440.9 1053.74   464.9 1041.66     493 1032.78
   505.2 1031.44     508 1031.60   634.4 1038.37   722.4 1052.12   769.1 1054.44
   828.7 1055.22   873.5 1060.70   931.9 1070.78  1043.9 1084.58  1065.6 1086.49
#Mann= 3 , 0 , 0
       0     0.1       0     493   0.045       0     508     0.1       0
Bank Sta=     493,     508
Exp/Cntr=0.3,0.1

Type RM Length L Ch R = 1 ,24322.1,398.297,413.447,408.061
XS GIS Cut Line= 3
     1753444.742      309243.766     1753503.684      309763.899
     1753899.864      310599.591
#Sta/Elev= 30
       0 1113.41    21.1 1108.17    48.2 1104.24    78.4 1093.34   102.6 1091.18
   117.9 1088.35   261.8 1082.90   286.0 1079.28   314.7 1072.21   374.5 1066.16
   431.0 1053.69   470.1 1039.84     516 1030.07   525.5 1028.75     531 1029.06
   632.8 1033.60   695.7 1031.71   714.4 1032.23   740.7 1041.34   753.8 1042.65
   808.9 1042.80   876.1 1045.76   937.7 1044.56   994.5 1051.27  1036.6 1054.16
  1176.3 1059.73  1292.5 1067.07  1371.3 1073.29  1435.5 1080.49  1448.3 1081.01
#Mann= 3 , 0 , 0
       0     0.1       0     516   0.045       0     531     0.1       0
#XS Ineff= 2 , 0
                          630.65         1033.71
Permanent Ineff=
       F       F
Bank Sta=     516,     531
Exp/Cntr=0.3,0.1

Type RM Length L Ch R = 1 ,23908.7,332.005,316.871,309.138
XS GIS Cut Line= 3
     1752967.436      309557.050     1753219.488      309987.589
     1753562.492      310478.880
#Sta/Elev= 30
       0 1155.36    35.3 1156.82    40.6 1156.51    52.6 1155.69    70.0 1150.87
   138.8 1106.83   160.5 1095.76   221.9 1066.38   278.2 1044.36   314.8 1031.81
   356.6 1029.41   452.2 1026.95   495.6 1026.76   510.6 1026.60   526.4 1026.28
   547.3 1026.86   559.3 1026.41   568.1 1027.06   575.4 1028.94   603.4 1040.55
   606.1 1041.24   674.3 1047.46   817.2 1049.96   878.5 1055.76   938.6 1058.00
   964.2 1060.14   996.0 1066.94  1047.7 1069.57  1075.1 1074.87  1097.9 1076.55
#Mann= 3 , 0 , 0
       0     0.1       0   495.6   0.045       0   510.6     0.1       0
Bank Sta=   495.6,   510.6
Exp/Cntr=0.3,0.1

Type RM Length L Ch R = 1 ,23591.8,365.555,362.672,355.713
XS GIS Cut Line= 3
     1752797.957      309653.832     1753021.618      310150.880
     1753384.334      310504.285
#Sta/Elev= 30
       0 1138.15    73.5 1137.78    93.0 1135.16   127.4 1125.53   142.6 1118.03
   199.2 1084.62   207.2 1080.50   253.1 1062.10   260.5 1058.64   301.3 1041.94
   322.9 1033.74   335.9 1030.79   481.2 1026.46   532.9 1026.18   547.9 1026.10
   603.9 1025.64   725.4 1025.87   736.5 1026.45   748.1 1029.78   750.6 1030.91
   757.8 1035.08   773.7 1045.41   782.1 1047.54   786.2 1048.33   811.6 1049.82
   857.9 1059.30   889.9 1064.17   985.1 1075.31  1024.5 1083.10  1051.5 1087.94
#Mann= 3 , 0 , 0
       0     0.1       0   532.9   0.045       0   547.9     0.1       0
Bank Sta=   532.9,   547.9
Exp/Cntr=0.3,0.1

Type RM Length L Ch R = 1 ,23229.1,399.855,400,391.739
XS GIS Cut Line= 3
     1752545.347      309727.553     1752752.591      310189.551
     1752910.249      310691.244
#Sta/Elev= 30
       0 1118.54    19.3 1117.90    78.9 1114.29    92.1 1111.74   137.8 1095.40
   148.0 1090.95   179.1 1080.16   208.9 1068.04   219.9 1064.27   241.9 1058.57
   294.0 1054.11   305.1 1053.69   327.4 1054.55   352.6 1052.62   392.6 1044.95
   435.9 1030.86   442.5 1029.51   461.8 1027.12   498.9 1025.27   506.3 1024.85
   513.9 1024.90   617.1 1024.88   751.3 1026.03   776.1 1030.32   793.0 1034.11
   847.5 1044.81   871.5 1046.13   897.1 1049.23   975.7 1061.91  1032.2 1074.12
#Mann= 3 , 0 , 0
       0     0.1       0   498.9   0.045       0   513.9     0.1       0
Bank Sta=   498.9,   513.9
Exp/Cntr=0.3,0.1

Type RM Length L Ch R = 1 ,22829.1,402.013,400,394.891
XS GIS Cut Line= 3
     1752154.554      309957.646     1752428.389      310373.498
     1752762.809      310765.351
#Sta/Elev= 30
       0 1104.78    23.9 1100.50    48.1 1093.96    66.8 1086.03    74.1 1085.29
    88.3 1088.60   109.6 1097.99   118.8 1099.31   149.7 1098.88   163.6 1099.50
   215.1 1099.48   252.0 1096.90   264.4 1095.13   314.7 1086.56   389.4 1069.88
   415.3 1062.25   435.3 1055.82   452.5 1048.45   474.7 1034.16   482.7 1028.22
   490.4 1024.21   502.8 1022.20   505.4 1022.24   698.1 1024.31   743.2 1029.49
   781.7 1032.12   810.0 1033.06   837.7 1037.72   934.0 1049.55  1013.1 1067.48
#Mann= 3 , 0 , 0
       0     0.1       0   490.4   0.045       0   505.4     0.1       0
Bank Sta=   490.4,   505.4
Exp/Cntr=0.3,0.1

Type RM Length L Ch R = 1 ,22429.1,404.379,400,397.75
XS GIS Cut Line= 3
     1751851.889      310252.768     1752154.605      310650.794
     1752555.697      310968.599
#Sta/Elev= 30
       0 1059.35    19.7 1058.33    38.4 1058.73    99.5 1062.44   167.8 1064.38
   215.4 1067.34   275.9 1067.05   317.1    1066   379.9 1062.11   393.1 1059.65
   401.8 1057.13   408.0 1054.78   435.7 1041.53   452.5 1029.95   464.4 1025.16
   492.6 1019.69   496.8 1019.13   507.6 1019.25   543.8 1019.81   630.0 1020.15
   689.5 1021.14   723.1 1021.31   753.7 1022.56   765.5 1024.67   781.4 1029.55
   792.4 1032.18   892.6 1049.27   917.6 1052.77   943.0 1054.24  1011.8 1068.53
#Mann= 3 , 0 , 0
       0     0.1       0   492.6   0.045       0   507.6     0.1       0
Bank Sta=   492.6,   507.6
Exp/Cntr=0.3,0.1

Type RM Length L Ch R = 1 ,22029.1,407.246,400,394.9
XS GIS Cut Line= 3
     1751569.463      310634.498     1751964.570      310984.579
     1752384.834      311247.379
#Sta/Elev= 30
       0 1165.72    10.6 1167.72    25.8 1168.69    84.4 1160.69   109.9 1155.02
   154.2 1134.53   187.3 1123.15   200.8 1117.77   221.7 1112.52   299.2 1103.93
   328.5 1099.43   346.8 1089.39   378.5 1067.70   404.2 1053.81   421.1 1042.29
   433.8 1035.12   441.9 1032.36   487.0 1021.35   517.1 1014.96   520.4 1014.85
   535.4 1014.34   545.7 1014.01   615.9 1016.09   708.0 1021.87   819.2 1032.03
   872.1 1041.30   900.7 1047.55   949.6 1053.18   969.4 1057.07  1023.6 1069.48
#Mann= 3 , 0 , 0
       0     0.1       0   520.4   0.045       0   535.4     0.1       0
Bank Sta=   520.4,   535.4
Exp/Cntr=0.3,0.1

Type RM Length L Ch R = 1 ,21629.1,404.23,400,396.725
XS GIS Cut Line= 3
     1751299.860      311144.473     1751809.119      311293.984
     1752283.793      311437.975
#Sta/Elev= 30
       0 1108.73    56.0 1091.69    72.2 1089.92   109.8 1089.12   201.6 1088.47
   262.8 1082.94   271.8 1080.92   285.3 1078.98   294.8 1075.20   338.7 1053.53
   382.1 1035.60   427.7 1025.59   436.4 1024.33   447.8 1024.42   452.7 1025.10
   464.9 1025.81   476.5 1021.97   493.5 1013.62   508.3 1011.38   516.7 1011.31
   523.3 1011.32   538.3 1011.35   555.5 1011.45   746.6 1015.68   776.8 1017.38
   882.6 1037.77   909.5 1041.21   933.7 1046.69   981.8 1061.15  1026.8 1073.28
#Mann= 3 , 0 , 0
       0     0.1       0   523.3   0.045       0   538.3     0.1       0
Bank Sta=   523.3,   538.3
Exp/Cntr=0.3,0.1

Type RM Length L Ch R = 1 ,21229.1,278.471,285.664,292.591
XS GIS Cut Line= 3
     1751206.422      311562.076     1751701.497      311650.485
     1752201.618      311735.530
#Sta/Elev= 30
       0 1198.79    17.3 1187.27    41.5 1175.71    76.9 1166.04    89.7 1160.11
   119.4 1137.96   152.5 1117.88   210.3 1085.98   222.4 1082.66   287.1 1083.29
   305.0 1080.68   337.4 1061.22   348.5 1058.24   380.9 1055.54   407.1 1047.37
   432.8 1034.89   465.7 1022.63   475.6 1019.96   486.2 1014.41   495.4 1012.16
   499.8 1010.39   510.4 1010.42   521.7 1010.39   707.7 1023.20   735.9 1024.15
   801.5 1030.97   836.5 1033.39   858.6 1037.79   943.5 1058.23  1010.2 1069.93
#Mann= 3 , 0 , 0
       0     0.1       0   495.4   0.045       0   510.4     0.1       0
Bank Sta=   495.4,   510.4
Exp/Cntr=0.3,0.1

Type RM Length L Ch R = 1 ,20943.5,615.804,606.628,595.789
XS GIS Cut Line= 3
     1751162.269      311668.977     1751618.733      311918.128
     1752058.959      312146.407
#Sta/Elev= 30
       0 1198.50     2.5 1197.60    24.2 1186.87   128.8 1126.73   144.1 1118.46
   173.9 1101.20   208.1 1086.41   223.3 1082.66   282.0 1080.89   299.1 1078.94
   329.2 1064.66   347.2 1058.24   391.7 1045.76   480.2 1019.38   502.6 1010.82
   511.3 1010.65   526.3 1010.29   529.5 1010.09   603.0 1010.10   629.0 1011.19
   695.7 1015.81   699.9 1016.45   761.7 1035.61   783.1 1037.67   798.3 1040.81
   826.0 1047.93   890.3 1060.42   966.0 1072.50   985.6 1076.58  1015.9 1079.76
#Mann= 3 , 0 , 0
       0     0.1       0   511.3   0.045       0   526.3     0.1       0
Bank Sta=   511.3,   526.3
Exp/Cntr=0.3,0.1

Type RM Length L Ch R = 1 ,20336.8,345.556,350.804,353.499
XS GIS Cut Line= 3
     1750962.543      312336.381     1751575.400      312382.402
     1752086.101      312391.687
#Sta/Elev= 30
       0 1029.10    22.1 1029.95    37.0 1031.64    52.4 1029.87    75.7 1028.46
   101.8 1025.70   199.1 1022.48   203.5 1021.97   246.1 1021.09   272.8 1018.08
   400.6 1012.27   544.9 1006.58   603.9 1006.42   612.9 1006.35   618.9 1006.85
   630.2 1011.36   654.5 1025.59   678.2 1038.32   683.4 1040.30   697.4 1042.27
   727.2 1044.92   828.5 1069.91   855.5 1075.39   903.8 1083.63   917.0 1085.37
   949.2 1088.28   963.7 1090.55   998.8 1101.66  1057.5 1116.60  1125.4 1127.56
#Mann= 3 , 0 , 0
       0     0.1       0   603.9   0.045       0   618.9     0.1       0
Bank Sta=   603.9,   618.9
Exp/Cntr=0.3,0.1

Type RM Length L Ch R = 1 ,19986,366.588,356.904,347.683
XS GIS Cut Line= 3
     1750929.979      312514.875     1751442.309      312623.824
     1751957.674      312711.787
#Sta/Elev= 30
       0 1069.96    56.6 1070.41    80.8 1069.82   147.3 1064.85   160.6 1062.44
   174.9 1060.76   215.1 1049.45   244.1 1040.61   262.8 1033.79   300.1 1017.25
   313.5 1014.27   415.6 1008.40   513.0 1003.84   518.3 1003.85   533.3 1003.92
   561.4 1005.65   574.5 1010.59   601.1 1024.60   612.5 1026.53   627.0 1027.27
   673.3 1038.77   735.3 1052.29   757.9 1057.99   802.4 1072.30   824.7 1075.55
   843.1 1076.58   874.1 1081.66   961.1 1105.66  1008.0 1117.67  1046.6 1130.55
#Mann= 3 , 0 , 0
       0     0.1       0   518.3   0.045       0   533.3     0.1       0
Bank Sta=   518.3,   533.3
Exp/Cntr=0.3,0.1

Type RM Length L Ch R = 1 ,19629.1,387.295,400,417.466
XS GIS Cut Line= 3
     1750913.037      313063.337     1751451.801      312905.201
     1751940.629      312735.250
#Sta/Elev= 30
       0 1097.71    27.4 1087.09    41.7 1082.35    80.6 1067.68    88.5 1065.69
   111.4 1064.22   150.8 1063.05   162.7 1061.41   207.2 1041.50   257.2 1022.24
   288.8 1011.95   311.2 1006.93   343.5 1005.89   441.5 1005.79     554 1002.33
   555.6 1002.29   564.7 1003.41     569 1003.46   607.1 1016.45   634.6 1018.62
   661.0 1025.55   690.3 1031.69   783.7 1053.64   815.0 1061.43   882.4 1076.81
   934.8 1085.21   998.5 1102.27  1007.5 1105.08  1049.8 1116.07  1079.0 1125.50
#Mann= 3 , 0 , 0
       0     0.1       0     554   0.045       0     569     0.1       0
Bank Sta=     554,     569
Exp/Cntr=0.3,0.1

Type RM Length L Ch R = 1 ,19229.1,404.741,400,389.134
XS GIS Cut Line= 3
     1750876.936      313083.431     1751349.682      313251.063
     1751812.326      313490.271
#Sta/Elev= 30
       0 1113.58    19.9 1105.27   104.9 1074.28   122.1 1066.97   140.8 1061.85
   159.3 1060.57   203.9 1060.16   216.5 1058.08   233.6 1051.63   254.3 1047.28
   279.5 1039.84   292.1 1031.68   298.7 1024.86   317.3 1010.55   324.9 1009.23
   341.8 1008.24   424.5 1005.77   471.6 1000.37   494.1  998.36   503.2  997.61
   509.1  998.42   542.1 1002.27   650.5 1006.48   689.7 1007.47   800.6 1012.91
   836.7 1014.04   851.9 1015.17   889.6 1014.54   916.6 1015.41  1022.4 1021.56
#Mann= 3 , 0 , 0
       0     0.1       0   494.1   0.045       0   509.1     0.1       0
Bank Sta=   494.1,   509.1
Exp/Cntr=0.3,0.1

Type RM Length L Ch R = 1 ,18829.1,401.461,400,404.168
XS GIS Cut Line= 3
     1750743.192      313538.788     1751231.503      313610.696
     1751771.154      313619.910
#Sta/Elev= 30
       0 1122.84    21.5 1117.89    69.8 1101.10    79.9 1096.73   105.0 1088.63
   142.8 1080.27   209.5 1062.55   220.0 1058.59   238.9 1048.14   257.5 1041.76
   279.7 1036.02   305.5 1031.73   332.5 1025.28   353.5 1018.52   364.1 1016.55
   407.7 1010.37   429.3 1009.03   449.8 1006.27   486.1  993.82   498.7  992.65
   501.1  992.85   594.7 1000.07   668.6 1002.82   755.3 1002.81   770.6 1004.59
   806.6 1018.62   829.9 1021.73   877.1 1030.74   972.4 1040.80  1033.3 1039.63
#Mann= 3 , 0 , 0
       0     0.1       0   486.1   0.045       0   501.1     0.1       0
Bank Sta=   486.1,   501.1
Exp/Cntr=0.3,0.1

Type RM Length L Ch R = 1 ,18429.1,295.193,294.263,294.016
XS GIS Cut Line= 3
     1750779.801      313939.858     1751286.691      313983.368
     1751777.355      314083.457
#Sta/Elev= 30
       0 1101.19    64.5 1085.04    89.7 1076.64   147.4 1055.27   160.3 1051.48
   188.2 1042.14   262.4 1023.84   292.5 1015.67   323.0 1006.91   338.1 1004.18
   360.3 1002.01   501.3  992.02   501.7  991.99   516.3  994.05   533.4 1003.31
   554.4 1008.67   637.9 1027.78   673.0 1034.53   698.7 1037.13   708.2 1040.05
   745.8 1054.99   772.1 1058.23   792.8 1062.52   814.7 1068.50   833.2 1072.15
   861.9 1080.14   892.6 1087.90   922.5 1093.63   986.9 1102.55  1009.5 1103.36
#Mann= 3 , 0 , 0
       0     0.1       0   501.3   0.045       0   516.3     0.1       0
Bank Sta=   501.3,   516.3
Exp/Cntr=0.3,0.1

Type RM Length L Ch R = 1 ,18134.9,489.204,505.736,519.339
XS GIS Cut Line= 3
     1750737.317      314237.506     1751247.314      314270.448
     1751740.804      314369.400
#Sta/Elev= 30
       0 1073.72    13.9 1069.88    66.4 1047.65    78.1 1043.83   122.3 1033.45
   187.9 1020.17   298.2 1005.59   325.1 1004.60   363.3 1004.94   376.0 1003.93
   387.6 1000.97   403.9  995.85   426.0  993.01   502.5  989.84   510.6  989.50
   517.5  990.10   605.4  998.77   628.0 1003.61   668.4 1014.47   689.6 1015.38
   705.8 1015.31   742.5 1021.79   795.5 1028.83   823.5 1033.14   844.8 1035.09
   888.8 1043.44   915.0 1047.52   938.6 1052.59   981.1 1065.52  1014.4 1076.35
#Mann= 3 , 0 , 0
       0     0.1       0   502.5   0.045       0   517.5     0.1       0
Bank Sta=   502.5,   517.5
Exp/Cntr=0.3,0.1

Type RM Length L Ch R = 1 ,17629.1,399.553,400,399.904
XS GIS Cut Line= 3
     1750682.326      314329.106     1751051.160      314684.471
     1751402.964      315037.566
#Sta/Elev= 30
       0 1062.06    30.2 1051.36    47.0 1044.74    68.7 1039.48   173.6 1022.68
   214.9 1017.67   294.3 1006.49   330.0 1002.33   339.3 1000.68   359.6  994.16
   372.3  991.57   406.6  987.34   504.7  986.10   515.4  986.02   519.7  986.90
   542.4  995.79   568.3  998.39   607.5 1010.85   643.1 1025.09   697.9 1043.80
   710.3 1049.17   732.2 1060.39   752.3 1071.57   794.3 1086.06   857.2 1102.04
   889.7 1109.34   940.0 1121.79   988.8 1127.60   999.9 1128.15  1010.6 1127.76
#Mann= 3 , 0 , 0
       0     0.1       0   504.7   0.045       0   519.7     0.1       0
Bank Sta=   504.7,   519.7
Exp/Cntr=0.3,0.1

Type RM Length L Ch R = 1 ,17229.1,398.082,400,404.715
XS GIS Cut Line= 3
     1750384.525      314572.673     1750737.558      314927.457
     1751091.907      315280.921
#Sta/Elev= 30
       0 1107.77    25.2 1102.92   100.7 1083.67   112.2 1080.02   150.3 1065.49
   179.8 1057.11   201.7 1047.68   271.1 1020.91   320.4 1005.34   334.1 1001.65
   346.0 1000.67   421.1 1000.18   454.7  995.34   471.5  991.41     493  982.46
   496.7  981.31     508  981.56   513.5  981.68   530.8  984.30   583.5  988.84
   617.2  994.27   640.7  999.40   679.0 1009.92   753.4 1027.21   784.4 1033.03
   834.7 1037.51   874.1 1039.11   897.6 1041.99   941.2 1044.47  1001.0 1045.38
#Mann= 3 , 0 , 0
       0     0.1       0     493   0.045       0     508     0.1       0
Bank Sta=     493,     508
Exp/Cntr=0.3,0.1

Type RM Length L Ch R = 1 ,16829.1,387.954,400,406.44
XS GIS Cut Line= 4
     1750146.511      314833.512     1750479.537      315228.554
     1750604.526      315419.156     1750580.888      315623.516
#Sta/Elev= 30
       0 1137.72    24.9 1125.43    48.8 1115.44    69.4 1105.50    80.7 1101.89
   130.5 1090.13   261.2 1039.72   270.4 1036.76   346.6 1014.48   398.4  998.08
   447.1  984.21   489.6  978.25   509.2  976.51   520.3  975.99   524.2  976.36
   592.8  982.81   615.5  984.05   660.9  988.19   688.7  989.62   708.7  993.88
   716.8  998.45   730.4 1003.53   744.6 1005.72   759.0 1009.38   778.4 1011.89
   814.1 1014.72   852.5 1013.55   879.5 1011.51   938.2 1010.89   950.3 1010.06
#Mann= 3 , 0 , 0
       0     0.1       0   509.2   0.045       0   524.2     0.1       0
Bank Sta=   509.2,   524.2
Exp/Cntr=0.3,0.1

Type RM Length L Ch R = 1 ,16429.1,411.9,400,394.244
XS GIS Cut Line= 3
     1750043.613      314887.063     1750135.110      315427.551
     1750277.884      315898.216
#Sta/Elev= 30
       0 1162.59    24.3 1152.76    38.3 1145.73    76.2 1129.07   102.2 1118.23
   119.0 1112.43   143.6 1102.98   156.8 1098.53   173.7 1092.01   189.8 1087.35
   251.3 1061.53   270.9 1054.73   336.0 1026.70   361.5 1011.49   397.6  987.44
   412.0  979.42   423.4  976.83   540.7  974.99   555.7  975.51   669.3  979.70
   728.0  983.96   752.9  984.15   788.1  983.65   816.3  987.06   827.3  989.11
   864.2  998.72   902.0 1002.68   929.9 1006.89   980.3 1014.91  1040.0 1025.53
#Mann= 3 , 0 , 0
       0     0.1       0   540.7   0.045       0   555.7     0.1       0
Bank Sta=   540.7,   555.7
Exp/Cntr=0.3,0.1

Type RM Length L Ch R = 1 ,16029.1,402.835,400,394.257
XS GIS Cut Line= 3
     1749486.086      315134.625     1749815.665      315536.020
     1750073.209      315961.252
#Sta/Elev= 30
       0 1087.43    25.3 1086.32    68.9 1082.72    89.5 1077.47   110.1 1073.43
   125.5 1064.19   134.4 1054.97   156.2 1035.50   171.6 1029.26   186.9 1028.71
   325.0 1032.95   341.1 1029.67   392.3 1008.72   417.0  996.71   446.8  983.12
   455.6  979.75   476.7  974.99   511.9  970.26   518.8  969.33   521.0  969.63
   526.9  971.69   544.8  977.53   552.1  978.10   574.7  978.90   795.2  982.89
   864.5  999.54   884.2 1001.29   907.8 1004.97  1004.2 1023.58  1016.5 1026.48
#Mann= 3 , 0 , 0
       0     0.1       0   511.9   0.045       0   526.9     0.1       0
Bank Sta=   511.9,   526.9
Exp/Cntr=0.3,0.1

Type RM Length L Ch R = 1 ,15629.1,322.578,310.884,303.283
XS GIS Cut Line= 3
     1749104.685      315380.946     1749465.425      315722.363
     1749842.607      316090.338
#Sta/Elev= 30
       0 1050.62     7.5 1048.53    24.2 1033.46    40.2 1022.86    49.4 1020.97
    72.9 1020.32    92.1 1021.41   171.0 1022.51   187.4 1019.12   220.0 1004.75
   245.0  999.30   271.3  992.19   309.8  983.26   335.5  979.53   341.8  979.67
   364.6  977.45   442.4  973.81   489.2  970.38   502.9  969.32   504.2  969.66
   518.0  973.24   538.8  976.39   746.8  974.71   780.0  975.72   786.7  977.09
   825.0  991.38   839.1  995.34   861.9  997.37   881.0 1000.68  1023.6 1029.27
#Mann= 3 , 0 , 0
       0     0.1       0   489.2   0.045       0   504.2     0.1       0
Bank Sta=   489.2,   504.2
Exp/Cntr=0.3,0.1

Type RM Length L Ch R = 1 ,15318.2,276.702,282.735,281.816
XS GIS Cut Line= 3
     1748805.650      315860.737     1749288.079      315966.595
     1749785.503      316186.287
#Sta/Elev= 30
       0 1146.32    14.9 1141.10    25.9 1135.61   152.2 1069.30   179.4 1053.52
   219.5 1025.13   224.1 1023.25   232.4 1020.61   348.2 1021.19   355.4 1019.96
   360.4 1018.48   368.6 1013.73   421.2  977.66   425.2  975.55   433.3  972.53
   445.2  971.16   489.1  969.72   504.1  969.08   507.1  968.95   594.7  977.75
   697.0  985.61   746.7  991.05   765.0  992.46   783.0  992.81   819.4  998.19
   934.8 1017.08   974.3 1027.41   998.4 1032.32  1008.1 1033.99  1037.7 1037.53
#Mann= 3 , 0 , 0
       0     0.1       0   489.1   0.045       0   504.1     0.1       0
Bank Sta=   489.1,   504.1
Exp/Cntr=0.3,0.1

Type RM Length L Ch R = 1 ,15035.5,714.443,717.12,722.193
XS GIS Cut Line= 3
     1748766.192      315954.297     1749210.700      316220.398
     1749697.532      316422.844
#Sta/Elev= 30
       0 1147.41    17.3 1143.69    26.9 1141.15    36.4 1137.24    48.3 1133.25
   193.3 1057.68   250.1 1024.18   264.4 1019.84   376.2 1017.29   388.5 1013.69
   431.7  990.62   458.3  977.18   468.3  974.34   497.8  969.96   516.2  967.91
   523.7  967.11   531.2  967.53   550.6  968.48   675.1  979.53   705.0  981.41
   715.1  985.16   733.8  990.39   761.7  994.07   805.3 1006.43   853.8 1011.49
   872.1 1015.23   932.2 1029.51   954.9 1034.39  1002.2 1048.21  1045.1 1058.69
#Mann= 3 , 0 , 0
       0     0.1       0   516.2   0.045       0   531.2     0.1       0
Bank Sta=   516.2,   531.2
Exp/Cntr=0.3,0.1

Type RM Length L Ch R = 1 ,14318.4,293.459,289.261,290.359
XS GIS Cut Line= 3
     1748451.333      316130.220     1748882.971      316409.065
     1749398.260      316804.921
#Sta/Elev= 30
       0 1134.72    35.2 1132.13    75.1 1124.17   115.8 1109.14   154.2 1093.29
   204.8 1075.01   240.7 1074.08   332.0 1078.36   346.2 1077.11   391.3 1061.18
   455.6 1032.80   539.0  967.48   543.1  965.71   547.4  963.92   555.9  963.28
   558.1  963.58   593.0  968.08   641.3  968.34   665.6  970.38   736.9  973.87
   830.3  984.38   843.8  983.73   860.2  974.84   871.8  979.38   875.2  979.76
   891.8  992.45   895.3  993.93   922.5  997.07  1000.0 1008.98  1163.7 1026.42
#Mann= 3 , 0 , 0
       0     0.1       0   543.1   0.045       0   558.1     0.1       0
Bank Sta=   543.1,   558.1
Exp/Cntr=0.3,0.1

Type RM Length L Ch R = 1 ,14029.1,408.803,400,389.973
XS GIS Cut Line= 3
     1748315.192      316447.701     1748739.962      316662.606
     1749228.970      317074.105
#Sta/Elev= 30
       0 1090.35    66.5 1067.57    85.6 1062.81   122.3 1055.02   146.1 1051.73
   163.6 1051.19   199.0 1051.49   233.2 1047.73   243.2 1047.38   265.6 1042.83
   366.9 1010.89   384.6 1003.43   405.2  990.49   430.6  972.85   443.3  967.90
   468.5  963.43   480.1  962.51   483.5  962.77   535.2  967.35   683.7  974.54
   773.6  985.05   841.7  990.67   847.5  992.00   898.9  999.62   919.4 1002.01
  1004.8 1015.13  1021.9 1017.11  1062.6 1015.82  1104.5 1012.04  1115.1 1012.57
#Mann= 3 , 0 , 0
       0     0.1       0   468.5   0.045       0   483.5     0.1       0
Bank Sta=   468.5,   483.5
Exp/Cntr=0.3,0.1

Type RM Length L Ch R = 1 ,13629.1,388.187,400,403.201
XS GIS Cut Line= 3
     1748156.355      316986.397     1748689.153      317032.493
     1749193.180      317168.826
#Sta/Elev= 30
       0 1148.68    22.1 1146.74    87.9 1146.34    93.5 1145.75   108.8 1141.24
   111.3 1140.92   117.8 1137.28   137.5 1127.96   275.2 1058.97   301.9 1048.28
   333.7 1034.51   373.2 1015.58   387.8 1009.10   411.5  997.18   421.1  991.85
   444.9  975.90   456.9  969.76   480.7  964.00   527.3  961.26   540.4  960.50
   542.3  960.68   658.8  974.04   708.1  978.75   731.1  980.14   847.9 1001.62
   862.3 1004.74   919.9 1012.04   974.9 1024.10  1026.4 1029.85  1056.9 1031.20
#Mann= 3 , 0 , 0
       0     0.1       0   527.3   0.045       0   542.3     0.1       0
Bank Sta=   527.3,   542.3
Exp/Cntr=0.3,0.1

Type RM Length L Ch R = 1 ,13229.1,388.79,400,414.299
XS GIS Cut Line= 3
     1748122.458      317090.905     1748608.662      317405.403
     1749058.925      317590.009
#Sta/Elev= 30
       0 1144.53    30.9 1142.06    48.0 1137.81   109.0 1108.01   153.4 1085.15
   219.7 1057.03   271.2 1038.49   313.8 1020.79   342.1 1003.21   357.1  996.69
   391.4  995.49   408.6  994.25   418.6  992.53   484.3  969.40   500.1  965.67
   571.6  959.15   582.1  958.55   586.6  958.97   660.0  970.41   690.5  972.77
   737.4  989.45   761.8 1000.70   775.7 1004.65   805.1 1009.01   840.3 1016.97
   883.7 1030.64   925.6 1047.43   968.2 1061.05  1041.1 1075.30  1065.7 1081.84
#Mann= 3 , 0 , 0
       0     0.1       0   571.6   0.045       0   586.6     0.1       0
Bank Sta=   571.6,   586.6
Exp/Cntr=0.3,0.1

Type RM Length L Ch R = 1 ,12829.1,405.297,400,390.181
XS GIS Cut Line= 3
     1748039.737      317162.655     1748308.189      317644.725
     1748569.040      318064.208
#Sta/Elev= 30
       0 1140.40    19.8 1138.31    56.8 1132.23    74.3 1125.23   134.5 1091.39
   150.8 1081.55   219.9 1051.47   249.2 1040.55   311.7 1018.95   322.3 1014.20
   331.4 1011.47   363.1 1004.16   407.3  997.93   413.9  996.36   464.8  973.96
   483.6  969.42   544.3  958.33   546.1  957.91   559.3  958.69   666.6  968.66
   675.0  968.92   683.7  970.55   692.3  975.27   718.1  996.18   735.4 1007.60
   744.0 1011.32   866.9 1050.28   910.9 1063.40   935.1 1069.50  1045.7 1093.72
#Mann= 3 , 0 , 0
       0     0.1       0   544.3   0.045       0   559.3     0.1       0
Bank Sta=   544.3,   559.3
Exp/Cntr=0.3,0.1

Type RM Length L Ch R = 1 ,12429.1,398.036,400,407.824
XS GIS Cut Line= 4
     1747619.789      317399.653     1747929.305      317740.120
     1748064.266      317866.471     1748496.881      318137.685
#Sta/Elev= 30
       0  991.31     4.7  992.07    27.0  991.51    40.9  992.49   117.3  991.96
   181.1  987.13   216.3  981.74   274.6  970.16   297.9  966.70   327.2  965.11
   409.3  963.33   481.7  960.59   586.3  960.06   637.5  956.83   646.2  956.07
   652.5  956.78   719.5  964.73   730.4  965.10   737.1  966.49   758.4  968.12
   772.4  972.55   785.1  980.73   800.4  987.99   835.9  998.63   880.9 1014.86
   906.8 1020.86   991.8 1048.06  1019.5 1055.02  1044.4 1059.86  1155.6 1079.21
#Mann= 3 , 0 , 0
       0     0.1       0   637.5   0.045       0   652.5     0.1       0
Bank Sta=   637.5,   652.5
Exp/Cntr=0.3,0.1

Type RM Length L Ch R = 1 ,12029.1,717.678,700.126,682.039
XS GIS Cut Line= 3
     1747378.367      317594.648     1747764.768      318093.603
     1748075.780      318503.200
#Sta/Elev= 30
       0 1027.74     8.2 1027.11    31.4 1023.15    66.3 1013.32   102.5  996.94
   135.5  979.94   151.2  972.81   160.4  970.37   260.4  962.09   324.2  957.73
   473.1  956.35   505.1  955.66   534.6  953.75   574.1  954.44   623.6  953.23
   624.8  953.20   638.6  954.20   665.6  962.57   692.6  965.83   715.9  979.19
   726.5  986.29   734.6  989.12   809.1 1007.07   868.7 1016.84   931.8 1029.79
   999.0 1045.46  1017.8 1050.94  1048.8 1062.13  1095.6 1075.44  1145.4 1091.19
#Mann= 3 , 0 , 0
       0     0.1       0   623.6   0.045       0   638.6     0.1       0
Bank Sta=   623.6,   638.6
Exp/Cntr=0.3,0.1

Type RM Length L Ch R = 1 ,11329,501.978,499.875,493.322
XS GIS Cut Line= 3
     1746959.258      318525.656     1747460.359      318459.865
     1747964.365      318542.068
#Sta/Elev= 30
       0  995.83    49.9  994.75    73.8  994.75    80.6  995.33   101.7  994.81
   122.9  991.10   150.4  984.80   175.3  976.99   181.6  975.59   258.0  963.02
   334.6  954.49   350.2  953.20   397.1  952.60   429.5  953.49   492.6  952.77
   513.8  952.01   516.9  951.89   528.8  952.77   602.7  958.16   616.7  958.74
   625.2  960.76   649.3  976.90   673.3  985.41   746.2 1006.92   836.1 1030.43
   870.8 1036.32   898.2 1042.00   938.0 1051.98   989.8 1068.70  1016.1 1076.39
#Mann= 3 , 0 , 0
       0     0.1       0   513.8   0.045       0   528.8     0.1       0
Bank Sta=   513.8,   528.8
Exp/Cntr=0.3,0.1

Type RM Length L Ch R = 1 ,10829.1,394.325,400,405.591
XS GIS Cut Line= 3
     1747020.980      318959.676     1747530.302      318950.749
     1748032.209      318893.772
#Sta/Elev= 30
       0 1056.61    24.1 1047.06    66.5 1031.88   108.3 1020.15   120.8 1017.07
   168.7 1001.82   249.0  982.64   272.7  975.80   282.5  972.41   314.6  958.34
   332.1  956.32   402.9  951.59   443.1  949.59   501.9  947.83   516.9  947.40
   517.5  947.38   527.7  949.57   542.5  951.10   560.3  954.68   573.4  955.18
   593.8  958.31   606.6  963.68   737.2 1023.78   749.1 1029.63   836.5 1068.33
   870.8 1079.63   935.3 1103.06   995.6 1123.29  1006.2 1125.83  1014.5 1127.24
#Mann= 3 , 0 , 0
       0     0.1       0   501.9   0.045       0   516.9     0.1       0
Bank Sta=   501.9,   516.9
Exp/Cntr=0.3,0.1

Type RM Length L Ch R = 1 ,10429.1,451.924,463.539,475.571
XS GIS Cut Line= 3
     1747030.434      319211.503     1747517.643      319323.535
     1748026.773      319384.330
#Sta/Elev= 30
       0 1069.72    56.0 1050.70    69.4 1046.95   105.2 1039.43   123.0 1034.88
   170.0 1026.10   277.6  990.32   290.2  984.10   294.4  981.29   325.5  957.67
   331.0  954.59   343.2  951.95   367.5  953.17   405.0  952.43   492.4  945.59
   501.5  945.08   507.4  946.26   516.7  947.04   531.5  950.65   561.3  953.83
   573.3  960.84   597.2  979.12   609.1  986.84   644.2  995.25   716.7 1020.99
   771.1 1039.41   863.1 1069.07   895.1 1073.21   970.4 1079.62  1012.7 1081.94
#Mann= 3 , 0 , 0
       0     0.1       0   492.4   0.045       0   507.4     0.1       0
Bank Sta=   492.4,   507.4
Exp/Cntr=0.3,0.1

Type RM Length L Ch R = 1 ,9965.6,340.924,342.874,347.889
XS GIS Cut Line= 3
     1747000.107      319330.987     1747461.936      319770.544
     1747885.972      320092.440
#Sta/Elev= 30
       0 1080.68    31.8 1071.89   106.4 1047.96   122.8 1045.28   147.5 1038.95
   270.7 1004.08   286.7  998.99   331.4  982.52   381.6  961.16   406.3  953.20
   487.2  947.69   531.0  945.60   609.6  945.32   631.6  944.20   634.1  944.35
   649.1  945.21   684.4  947.91   709.5  947.06   741.4  947.95   775.4  954.12
   798.9  955.10   806.9  956.48   845.8  969.16   927.7 1007.97   938.6 1011.46
  1048.2 1031.65  1068.8 1035.09  1094.3 1036.34  1129.6 1034.74  1169.9 1035.79
#Mann= 3 , 0 , 0
       0     0.1       0   634.1   0.045       0   649.1     0.1       0
Bank Sta=   634.1,   649.1
Exp/Cntr=0.3,0.1

Type RM Length L Ch R = 1 ,9622.7,401.622,393.586,387.48
XS GIS Cut Line= 3
     1746833.194      319456.522     1747163.152      319812.419
     1747541.295      320260.767
#Sta/Elev= 30
       0 1094.48    99.5 1069.72   141.5 1057.79   180.1 1042.55   220.2 1025.45
   259.3 1014.27   275.6 1007.97   318.7  988.31   374.8  971.43   435.3  956.42
   470.6  944.49   479.2  943.38   488.0  942.04   494.2  941.96   497.8  941.92
   553.2  945.08   648.7  947.43   791.1  947.93   867.0  949.56   881.3  951.40
   886.3  952.75   904.5  960.52   917.1  964.82   942.9  968.06   969.5  979.35
   980.2  984.53  1001.1  992.63  1041.7 1010.22  1049.4 1012.93  1071.8 1014.83
#Mann= 3 , 0 , 0
       0     0.1       0   479.2   0.045       0   494.2     0.1       0
Bank Sta=   479.2,   494.2
Exp/Cntr=0.3,0.1

Type RM Length L Ch R = 1 ,9229.1,360.109,362.979,367.719
XS GIS Cut Line= 3
     1746526.640      319926.145     1746980.767      320155.718
     1747393.273      320436.547
#Sta/Elev= 30
       0 1100.54    15.6 1099.89    77.4 1092.37    87.4 1090.68   128.9 1081.09
   137.0 1078.73   220.9 1051.44   270.6 1032.60   281.3 1029.31   320.3 1015.40
   357.2 1001.15   390.5  989.62   404.6  983.09   461.0  952.32   492.0  943.01
   501.4  940.95   502.1  940.80   516.4  940.96   568.9  943.50   663.1  946.96
   684.6  946.70   787.4  951.96   844.3  958.84   890.1  971.30   921.2  975.26
   924.2  976.35   944.8  988.43   958.4  997.55   974.8 1005.00  1007.9 1006.83
#Mann= 3 , 0 , 0
       0     0.1       0   501.4   0.045       0   516.4     0.1       0
Bank Sta=   501.4,   516.4
Exp/Cntr=0.3,0.1

Type RM Length L Ch R = 1 ,8866.1,430.886,437.021,438.919
XS GIS Cut Line= 3
     1746389.955      320182.785     1746833.619      320482.430
     1747147.964      320860.003
#Sta/Elev= 30
       0 1140.96    16.0 1134.48    50.0 1123.46   139.4 1101.83   161.1 1095.75
   169.2 1092.47   248.0 1048.61   277.4 1034.25   314.8 1020.44   374.1  997.08
   395.0  986.84   440.2  952.60   450.9  946.75   462.0  944.41   521.6  938.26
   521.9  938.27   536.9  938.65   681.1  943.66   727.5  948.31   757.0  952.87
   784.8  960.60   809.4  963.35   817.7  965.51   843.0  981.40   891.1  988.61
   945.0  999.67   957.5 1001.17   975.6 1004.92  1011.6 1009.38  1026.7 1012.15
#Mann= 3 , 0 , 0
       0     0.1       0   521.9   0.045       0   536.9     0.1       0
Bank Sta=   521.9,   536.9
Exp/Cntr=0.3,0.1

Type RM Length L Ch R = 1 ,8429.1,397.933,400,405.24
XS GIS Cut Line= 3
     1746220.035      320410.872     1746547.256      320787.286
     1746872.827      321181.399
#Sta/Elev= 30
       0 1142.54    27.4 1131.64    59.7 1122.32   187.4 1095.56   210.4 1083.75
   279.3 1043.37   295.8 1034.97   333.5 1021.05   380.3  999.19   421.1  976.07
   443.2  960.05   472.9  940.98   491.3  937.20   501.8  936.33   506.3  936.51
   587.5  940.72   686.3  944.05   712.1  943.24   787.9  945.87   798.4  948.20
   818.6  956.75   843.9  961.31   858.3  970.38   907.0 1004.98   921.6 1013.70
   933.0 1018.56   956.4 1026.08   977.1 1029.20   995.7 1029.60  1010.0 1033.33
#Mann= 3 , 0 , 0
       0     0.1       0   491.3   0.045       0   506.3     0.1       0
Bank Sta=   491.3,   506.3
Exp/Cntr=0.3,0.1

Type RM Length L Ch R = 1 ,8029.1,325.805,334.262,337.858
XS GIS Cut Line= 3
     1745919.437      320582.076     1746223.685      320982.016
     1746481.815      321429.337
#Sta/Elev= 30
       0 1098.09    20.1 1094.82    77.8 1076.03   155.6 1048.20   184.2 1037.56
   214.0 1028.32   224.7 1025.34   280.4 1007.62   365.3  978.33   417.5  958.67
   428.3  954.31   458.9  943.60   483.7  938.14   488.7  936.28     495  934.59
   503.7  933.67     510  933.89   609.5  937.29   782.0  948.43   814.2  950.91
   854.3  954.47   868.0  957.87   871.9  960.31   881.7  965.52   891.7  971.33
   932.9  983.11   957.0  989.08   977.6  993.42  1012.0  998.29  1019.0  998.76
#Mann= 3 , 0 , 0
       0     0.1       0     495   0.045       0     510     0.1       0
Bank Sta=     495,     510
Exp/Cntr=0.3,0.1

Type RM Length L Ch R = 1 ,7694.9,486.755,465.739,452.48
XS GIS Cut Line= 3
     1745813.510      320628.063     1745939.118      321126.223
     1746083.094      321614.134
#Sta/Elev= 30
       0 1085.93    20.9 1079.66    88.0 1054.56   110.1 1045.05   165.0 1017.12
   182.7 1010.26   212.3 1006.37   226.2 1003.69   236.1 1000.67   245.0  997.21
   275.1  988.26   360.9  955.15   373.0  952.20   406.1  947.12   428.9  944.62
   483.3  941.53   504.7  934.35   511.3  933.11   519.7  933.58   598.8  938.18
   685.2  938.22   757.5  943.25   860.0  953.68   865.0  955.44   940.3  993.17
   951.3  997.86   965.7 1001.86   981.3 1004.26  1004.5 1011.34  1022.5 1017.91
#Mann= 3 , 0 , 0
       0     0.1       0   504.7   0.045       0   519.7     0.1       0
Bank Sta=   504.7,   519.7
Exp/Cntr=0.3,0.1

Type RM Length L Ch R = 1 ,7229.1,397.172,400,398.552
XS GIS Cut Line= 3
     1745128.716      321153.324     1745585.572      321343.354
     1745999.495      321678.808
#Sta/Elev= 30
       0 1104.33    52.1 1092.24    90.8 1080.83   162.9 1056.87   195.9 1041.63
   287.9 1003.91   338.8  981.84   377.2  962.58   388.1  958.62   445.2  949.95
   462.6  943.99   487.3  931.34   495.2  929.80   502.3  930.46   542.7  934.19
   623.7  936.93   654.1  936.79   691.4  939.02   715.0  941.65   737.3  949.39
   768.9  952.53   777.3  955.22   807.9  967.42   858.3  990.96   875.4  996.80
   926.1 1003.86   976.7 1003.63   989.4 1004.42  1009.1 1007.09  1027.6 1012.80
#Mann= 3 , 0 , 0
       0     0.1       0   487.3   0.045       0   502.3     0.1       0
Bank Sta=   487.3,   502.3
Exp/Cntr=0.3,0.1

Type RM Length L Ch R = 1 ,6829.1,391.646,400,405.992
XS GIS Cut Line= 3
     1744983.393      321445.744     1745437.114      321704.616
     1745840.681      321993.808
#Sta/Elev= 30
       0 1082.93    80.0 1062.93   118.7 1050.46   180.7 1021.11   201.1 1013.17
   238.7 1001.36   274.2  987.92   293.6  982.08   309.5  977.52   338.3  971.04
   377.1  964.20   448.5  949.18   490.3  938.00   514.9  928.26   524.7  927.11
   529.9  927.93   541.7  930.19   557.0  931.10   563.1  930.77   732.3  935.50
   746.9  939.24   761.7  946.93   770.6  949.81   776.1  951.06   790.7  952.04
   804.9  956.16   840.3  973.95   883.4  987.32   955.2 1006.40  1018.9 1018.22
#Mann= 3 , 0 , 0
       0     0.1       0   514.9   0.045       0   529.9     0.1       0
Bank Sta=   514.9,   529.9
Exp/Cntr=0.3,0.1

Type RM Length L Ch R = 1 ,6429.1,399.945,400,401.326
XS GIS Cut Line= 3
     1744837.174      321595.612     1745153.164      321983.749
     1745469.154      322371.887
#Sta/Elev= 30
       0 1095.69    48.8 1082.59    54.6 1081.78    86.1 1075.60    97.2 1072.16
   103.6 1069.71   122.9 1060.85   137.5 1054.70   168.1 1039.49   188.4 1028.20
   218.1 1015.46   275.2  994.13   300.4  981.07   348.2  968.35   463.1  939.85
   488.9  929.76     493  928.90   502.9  926.70     508  927.01   573.5  930.73
   785.7  935.70   807.1  938.01   816.9  942.08   831.6  947.46   851.3  949.12
   864.2  953.42   936.8  995.33   968.7 1012.50   997.3 1023.73  1001.0 1024.89
#Mann= 3 , 0 , 0
       0     0.1       0     493   0.045       0     508     0.1       0
Bank Sta=     493,     508
Exp/Cntr=0.3,0.1

Type RM Length L Ch R = 1 ,6029.1,478.467,493.175,506.122
XS GIS Cut Line= 3
     1744556.997      321867.351     1744879.039      322267.493
     1745169.119      322672.299
#Sta/Elev= 30
       0 1085.20    47.2 1069.29    73.3 1055.65   101.1 1035.33   114.8 1028.61
   153.8 1013.96   214.7  997.69   230.1  992.23   274.8  982.40   340.6  971.07
   421.3  948.97   458.6  943.68   473.6  940.28   506.1  926.01   519.8  924.00
   521.1  924.03   630.1  925.56   680.0  927.96   718.8  932.48   740.3  937.52
   758.4  946.11   777.9  948.58   792.4  953.85   817.9  970.53   869.0  988.01
   898.7 1004.81   934.0 1027.22   969.7 1046.71   988.1 1050.70  1011.6 1053.63
#Mann= 3 , 0 , 0
       0     0.1       0   506.1   0.045       0   521.1     0.1       0
Bank Sta=   506.1,   521.1
Exp/Cntr=0.3,0.1

Type RM Length L Ch R = 1 ,5536,301.99,306.825,312.408
XS GIS Cut Line= 3
     1744456.709      321920.498     1744468.918      322435.474
     1744499.526      322960.668
#Sta/Elev= 30
       0 1078.59    19.0 1072.58   128.8 1028.48   227.0  991.07   240.2  987.16
   282.7  977.19   330.8  967.50   388.8  954.28   461.3  936.93   470.5  934.23
   474.4  932.28   478.3  931.21   496.4  924.37   500.3  923.29   506.1  923.19
   511.4  923.25   582.1  924.37   629.3  927.91   739.3  941.38   751.3  942.09
   759.1  943.49   770.4  944.66   775.4  947.50   783.2  950.98   815.3  970.93
   830.9  974.42   843.6  975.32   877.6  976.49   988.9  978.47  1041.2  979.88
#Mann= 3 , 0 , 0
       0     0.1       0   496.4   0.045       0   511.4     0.1       0
Bank Sta=   496.4,   511.4
Exp/Cntr=0.3,0.1

Type RM Length L Ch R = 1 ,5229.1,402.21,400,397.709
XS GIS Cut Line= 3
     1744266.885      321914.819     1744177.006      322411.273
     1744080.374      322914.597
#Sta/Elev= 30
       0 1089.68    63.6 1066.33   121.8 1043.35   222.7 1004.74   243.3  997.45
   274.4  985.30   311.2  975.84   338.7  969.38   376.2  961.10   420.5  949.16
   461.0  937.68   495.8  924.63     497  924.51   509.9  923.02     512  923.09
   692.3  929.22   702.7  930.89   744.1  945.23   768.7  947.37   785.8  952.84
   822.2  968.22   830.2  973.11   845.4  984.27   882.7 1013.79   890.9 1019.60
   914.1 1034.30   946.7 1051.95   951.5 1053.84   979.0 1060.17  1017.0 1067.26
#Mann= 3 , 0 , 0
       0     0.1       0     497   0.045       0     512     0.1       0
Bank Sta=     497,     512
Exp/Cntr=0.3,0.1

Type RM Length L Ch R = 1 ,4829.1,277.289,283.879,292.177
XS GIS Cut Line= 3
     1743850.290      321846.966     1743806.719      322347.828
     1743758.488      322856.239
#Sta/Elev= 30
       0 1086.51    22.0 1077.86    64.2 1062.38    93.2 1052.92   142.1 1035.57
   166.0 1027.62   216.1 1009.75   302.7  977.86   380.3  959.57   418.5  944.50
   437.4  940.43   469.8  934.22   495.3  924.52   498.2  923.41   510.3  923.03
   564.1  921.26   592.5  924.52   600.0  924.52   617.5  925.91   621.8  926.94
   643.6  934.01   676.2  938.29   687.7  942.84   778.8  989.71   789.2  995.67
   816.5 1012.70   852.2 1035.57   864.5 1041.36   916.1 1058.44  1013.4 1080.09
#Mann= 3 , 0 , 0
       0     0.1       0   495.3   0.045       0   510.3     0.1       0
Bank Sta=   495.3,   510.3
Exp/Cntr=0.3,0.1
